HEC-RAS study k145-00-00.prj: K145-00-00

--- k145-00-00.g01 (geometry) --- (continued)

Type RM Length L Ch R = 3 ,17419   ,,,
BEGIN DESCRIPTION:
CYPRESS CHASE DRIVE
Structure ID: K145-00-00-S8
END DESCRIPTION:
Bridge Culvert--1,0,-1,-1, 0
Deck Dist Width WeirC Skew NumUp NumDn MinLoCord MaxHiCord MaxSubmerge Is_Ogee
10,95,2.6,0, 60, 60, , , .95, 0, ,,,
 -4395.9 -3635.9 -3475.9 -3365.9 -3185.9 -3095.9 -2915.9 -2725.9 -2585.9 -2485.9
 -2245.9 -2015.9 -1975.9 -1915.9 -1755.9 -1605.9 -1535.9 -1475.9 -1435.9 -1105.9
  -795.9  -765.9  -725.9  -665.9  1754.1  1794.1  1974.1  2004.1  2214.1  2274.1
  2414.1  2444.1  2924.1  3024.1  3094.1  3204.1  3454.1  3634.1  3764.1  4114.1
  4254.1  4304.1  4494.1  4594.1  4919.2 4944.79  4944.9 4954.81  5044.9  5054.9
 5055.01  5570.3  5720.3  5840.3  6720.3  6760.3  6800.3  6850.3  6900.3  7006.9
   166.6   160.6   158.1   160.2   160.3   156.5   159.7   158.1   155.1   156.8
     157   155.7     154   156.2   154.5   155.7     154   155.2   153.9   152.7
     153   151.6   153.7   151.7     151   153.2   151.8   153.2   153.4   150.9
   152.7   150.8   149.8   151.3   149.6   151.8   150.3   152.5   151.2   153.6
   151.3   153.5   152.7   150.4   153.3  153.32  157.12  157.18   157.4  157.36
  153.56     150   149.9   153.1   151.2   153.2   149.1   149.7     154     154
   166.6   160.6   158.1   160.2   160.3   156.5   159.7   158.1   155.1   156.8
     157   155.7     154   156.2   154.5   155.7     154   155.2   153.9   152.7
     153   151.6   153.7   151.7     151   153.2   151.8   153.2   153.4   150.9
   152.7   150.8   149.8   151.3   149.6   151.8   150.3   152.5   151.2   153.6
   151.3   153.5   152.7   150.4  153.29  152.39  152.36  149.76  150.26  152.89
  152.92     150   149.9   153.1   151.2   153.2   149.1   149.7     154     154
 -4395.9 -3635.9 -3475.9 -3365.9 -3185.9 -3095.9 -2915.9 -2725.9 -2585.9 -2485.9
 -2245.9 -2015.9 -1975.9 -1915.9 -1755.9 -1605.9 -1535.9 -1475.9 -1435.9 -1105.9
  -795.9  -765.9  -725.9  -665.9  1754.1  1794.1  1974.1  2004.1  2214.1  2274.1
  2414.1  2444.1  2924.1  3024.1  3094.1  3204.1  3454.1  3634.1  3764.1  4114.1
  4254.1  4304.1  4494.1  4594.1  4919.2 4944.79  4944.9 4954.81  5044.9  5054.9
 5055.01  5570.3  5720.3  5840.3  6720.3  6760.3  6800.3  6850.3  6900.3  7006.9
   166.6   160.6   158.1   160.2   160.3   156.5   159.7   158.1   155.1   156.8
     157   155.7     154   156.2   154.5   155.7     154   155.2   153.9   152.7
     153   151.6   153.7   151.7     151   153.2   151.8   153.2   153.4   150.9
   152.7   150.8   149.8   151.3   149.6   151.8   150.3   152.5   151.2   153.6
   151.3   153.5   152.7   150.4   153.3  153.32  157.12  157.18   157.4  157.36
  153.56     150   149.9   153.1   151.2   153.2   149.1   149.7     154     154
   166.6   160.6   158.1   160.2   160.3   156.5   159.7   158.1   155.1   156.8
     157   155.7     154   156.2   154.5   155.7     154   155.2   153.9   152.7
     153   151.6   153.7   151.7     151   153.2   151.8   153.2   153.4   150.9
   152.7   150.8   149.8   151.3   149.6   151.8   150.3   152.5   151.2   153.6
   151.3   153.5   152.7   150.4  153.29  152.39  152.36  149.76  150.26  152.89
  152.92     150   149.9   153.1   151.2   153.2   149.1   149.7     154     154
Pier Skew, UpSta & Num, DnSta & Num=  ,4984.4, 2 ,4984.4, 2 , 0 , 0 , 0 ,,
     1.3     1.3
  141.78  151.85
     1.3     1.3
  142.32  152.39
Pier Skew, UpSta & Num, DnSta & Num=  ,5014.5, 2 ,5014.5, 2 , 0 , 0 , 0 ,,
     1.3     1.3
  141.01  151.94
     1.3     1.3
  141.55  152.48
BR Coef= 1 , 1 , 1 ,1.25, 0 ,,,.8,0,2,0,
WSPro=,,,, 1 ,,,, 0 ,,,, 0 ,,,,-1 ,-1 ,-1 , 0 , 0 , 0 , 0 , 0
BR U #Sta/Elev= 194
 -4395.9   166.6 -4305.9   166.6 -4295.9   165.9 -4095.9   164.7 -3775.9   160.9
 -3635.9   160.6 -3595.9   159.5 -3475.9   158.1 -3465.9   158.5 -3415.9   158.6
 -3365.9   160.2 -3295.9   160.1 -3285.9   160.5 -3185.9   160.3 -3095.9   156.5
 -3015.9   158.4 -3005.9   159.1 -2915.9   159.7 -2895.9   159.2 -2785.9   157.9
 -2755.9   158.2 -2725.9   158.1 -2695.9     157 -2665.9   156.3 -2585.9   155.1
 -2485.9   156.8 -2265.9   156.4 -2245.9     157 -2195.9   156.4 -2015.9   155.7
 -1985.9   154.2 -1975.9     154 -1915.9   156.2 -1805.9   155.2 -1785.9   154.7
 -1765.9   155.4 -1755.9   154.5 -1735.9   155.4 -1725.9   154.7 -1715.9   154.7
 -1705.9   155.2 -1685.9   154.9 -1675.9   155.6 -1665.9   155.1 -1625.9   155.7
 -1605.9   155.7 -1575.9   155.1 -1565.9   154.6 -1535.9     154 -1505.9   154.3
 -1495.9   153.9 -1475.9   155.2 -1445.9     154 -1435.9   153.9 -1425.9   154.4
 -1325.9   153.5 -1265.9   153.3 -1125.9   153.3 -1105.9   152.7 -1085.9   153.7
  -815.9   152.8  -795.9     153  -765.9   151.6  -725.9   153.7  -695.9   153.6
  -665.9   151.7  -615.9   152.4  -185.9   151.5   -95.9   151.4   -85.9   151.1
    84.1   151.5   584.1   151.6   844.1   151.4  1741.9   151.4  1744.1   151.4
  1754.1     151  1774.1   151.7  1784.1   152.7  1794.1   153.2  1904.1   152.8
  1944.1   151.8  1974.1   151.8  2004.1   153.2  2214.1   153.4  2224.1   153.1
  2254.1   151.1  2274.1   150.9  2354.1   152.5  2414.1   152.7  2444.1   150.8
  2894.1   150.6  2924.1   149.8  2927.8  149.95  2934.1   150.2  2944.1     151
  3024.1   151.3  3094.1   149.6  3114.1   150.8  3204.1   151.8  3214.1   151.6
  3234.1   151.8  3334.1   151.5  3364.1   151.8  3394.1   151.3  3414.1   151.3
  3454.1   150.3  3534.1   151.3  3584.1   152.1  3604.1   151.9  3634.1   152.5
  3764.1   151.2  3784.1   151.6  3928.5  151.74  3994.1   151.8  4044.1   152.2
  4114.1   153.6  4154.1   152.8  4168.2  152.59  4254.1   151.3  4304.1   153.5
  4494.1   152.7  4564.1   151.6  4594.1   150.4  4753.2  152.39    4775  152.66
  4824.8  152.88  4825.3  152.88  4875.7   153.1  4919.2  153.29    4921  153.26
  4942.6  152.96 4944.79  152.39  4944.9  152.36 4945.01  152.33  4954.7  149.79
 4954.81  149.76  4954.9  149.74  4955.7  149.53  4972.7  144.18  4984.3  142.99
  4984.4  142.95  4985.1  142.77  4991.2  141.22  4998.8  140.82  5005.5   140.9
  5008.8  141.24  5014.5  142.11  5015.1  142.22  5026.5  144.23  5043.9     150
 5044.69  150.21  5044.8  150.24  5044.9  150.26 5054.79  152.86  5054.9  152.89
 5055.01  152.92  5058.2  153.76  5094.8  153.59  5102.4  153.56  5144.1  153.02
  5196.6  152.33  5246.6  151.68  5500.3   151.1  5530.3   150.4  5550.3   150.1
  5560.3   150.4  5570.3     150  5618.7  150.36  5650.3   150.6  5720.3   149.9
  5760.3   151.6  5790.3     152  5800.3   152.4  5840.3   153.1  5850.3   152.9
  5950.3   152.9  6100.3   152.5  6190.3   151.5  6270.3   152.1  6380.3   151.2
  6720.3   151.2  6740.3   152.7  6750.3   153.2  6760.3   153.2  6780.3   151.2
  6790.3   149.7  6800.3   149.1  6830.3   149.7  6850.3   149.7  6860.3   150.3
  6880.3   152.8  6900.3     154  6950.3     155  7006.9     154
BR U #Mann= 3
 -4395.9     .99  4942.6     .04  5058.2     .99
BR U Banks=4942.6,5058.2
BR D #Sta/Elev= 194
 -4395.9   166.6 -4305.9   166.6 -4295.9   165.9 -4095.9   164.7 -3775.9   160.9
 -3635.9   160.6 -3595.9   159.5 -3475.9   158.1 -3465.9   158.5 -3415.9   158.6
 -3365.9   160.2 -3295.9   160.1 -3285.9   160.5 -3185.9   160.3 -3095.9   156.5
 -3015.9   158.4 -3005.9   159.1 -2915.9   159.7 -2895.9   159.2 -2785.9   157.9
 -2755.9   158.2 -2725.9   158.1 -2695.9     157 -2665.9   156.3 -2585.9   155.1
 -2485.9   156.8 -2265.9   156.4 -2245.9     157 -2195.9   156.4 -2015.9   155.7
 -1985.9   154.2 -1975.9     154 -1915.9   156.2 -1805.9   155.2 -1785.9   154.7
 -1765.9   155.4 -1755.9   154.5 -1735.9   155.4 -1725.9   154.7 -1715.9   154.7
 -1705.9   155.2 -1685.9   154.9 -1675.9   155.6 -1665.9   155.1 -1625.9   155.7
 -1605.9   155.7 -1575.9   155.1 -1565.9   154.6 -1535.9     154 -1505.9   154.3
 -1495.9   153.9 -1475.9   155.2 -1445.9     154 -1435.9   153.9 -1425.9   154.4
 -1325.9   153.5 -1265.9   153.3 -1125.9   153.3 -1105.9   152.7 -1085.9   153.7
  -815.9   152.8  -795.9     153  -765.9   151.6  -725.9   153.7  -695.9   153.6
  -665.9   151.7  -615.9   152.4  -185.9   151.5   -95.9   151.4   -85.9   151.1
    84.1   151.5   584.1   151.6   844.1   151.4  1741.9   151.4  1744.1   151.4
  1754.1     151  1774.1   151.7  1784.1   152.7  1794.1   153.2  1904.1   152.8
  1944.1   151.8  1974.1   151.8  2004.1   153.2  2214.1   153.4  2224.1   153.1
  2254.1   151.1  2274.1   150.9  2354.1   152.5  2414.1   152.7  2444.1   150.8
  2894.1   150.6  2924.1   149.8  2927.8  149.95  2934.1   150.2  2944.1     151
  3024.1   151.3  3094.1   149.6  3114.1   150.8  3204.1   151.8  3214.1   151.6
  3234.1   151.8  3334.1   151.5  3364.1   151.8  3394.1   151.3  3414.1   151.3
  3454.1   150.3  3534.1   151.3  3584.1   152.1  3604.1   151.9  3634.1   152.5
  3764.1   151.2  3784.1   151.6  3928.5  151.74  3994.1   151.8  4044.1   152.2
  4114.1   153.6  4154.1   152.8  4168.2  152.59  4254.1   151.3  4304.1   153.5
  4494.1   152.7  4564.1   151.6  4594.1   150.4  4753.2  152.39    4775  152.66
  4824.8  152.88  4825.3  152.88  4875.7   153.1  4919.2  153.29    4921  153.26
  4942.6  152.96 4944.79  152.93  4944.9   152.9 4945.01  152.87  4954.7  150.33
 4954.81   150.3  4954.9  150.28  4955.7  150.07  4972.7  144.72  4984.3  143.53
  4984.4  143.49  4985.1  143.31  4991.2  141.76  4998.8  141.36  5005.5  141.44
  5008.8  141.78  5014.5  142.65  5015.1  142.76  5026.5  144.77  5043.9  150.54
 5044.69  150.75  5044.8  150.78  5044.9   150.8 5054.79   153.4  5054.9  153.43
 5055.01  153.46  5058.2  153.76  5094.8  153.59  5102.4  153.56  5144.1  153.02
  5196.6  152.33  5246.6  151.68  5500.3   151.1  5530.3   150.4  5550.3   150.1
  5560.3   150.4  5570.3     150  5618.7  150.36  5650.3   150.6  5720.3   149.9
  5760.3   151.6  5790.3     152  5800.3   152.4  5840.3   153.1  5850.3   152.9
  5950.3   152.9  6100.3   152.5  6190.3   151.5  6270.3   152.1  6380.3   151.2
  6720.3   151.2  6740.3   152.7  6750.3   153.2  6760.3   153.2  6780.3   151.2
  6790.3   149.7  6800.3   149.1  6830.3   149.7  6850.3   149.7  6860.3   150.3
  6880.3   152.8  6900.3     154  6950.3     155  7006.9     154
BR D #Mann= 3
 -4395.9     .99  4942.6     .04  5058.2     .99
BR D Banks=4942.6,5058.2
BC Design=,, 0 ,, 0 ,,,,,,
BC HTab HWMax=166.6

Type RM Length L Ch R = 1 ,17306   ,97.85,100,102.3
BEGIN DESCRIPTION:
S8_CYPRESS CHASE DR-DS - XS2
END DESCRIPTION:
XS GIS Cut Line= 4
      3014564.41      13926787.2      3010745.99     13919098.01
      3010699.59     13918997.01       3009771.9     13917285.01
#Sta/Elev= 30
 -3635.9   160.6 -3475.9   158.1 -3185.9   160.3 -3095.9   156.5 -2915.9   159.7
 -2585.9   155.1 -2245.9     157 -1975.9     154 -1605.9   155.7  -765.9   151.6
  -725.9   153.7  1754.1     151  2214.1   153.4  2274.1   150.9  2414.1   152.7
  3094.1   149.6  4114.1   153.6  4594.1   150.4  4942.6  152.96  4972.7  144.69
  4998.8  141.33  5026.5  144.74  5058.2  153.76  5720.3   149.9  5840.3   153.1
  6720.3   151.2  6760.3   153.2  6800.3   149.1  6900.3     154  7006.9     154
#Mann= 3 ,-1 , 0
 -3635.9     .99       0  4942.6     .04       0  5058.2     .99       0
Levee=0,,,-1,5217,151.1,,
#XS Ineff= 2 , 0
       0    4944   151.6    5054       0   151.6
Permanent Ineff=
       F       F
#Block Obstruct= 1 ,-1
 2424.71    3650   151.3
Bank Sta=4942.6,5058.2
XS Rating Curve= 0
Exp/Cntr=.5,.3

Type RM Length L Ch R = 1 ,17206   ,598.84,612,626.1
BEGIN DESCRIPTION:
S8_CYPRESS CHASE DR-DS - XS1
END DESCRIPTION:
XS GIS Cut Line= 4
      3014571.77      13926776.5      3010839.12     13919056.42
      3010792.71     13918955.42      3009865.03     13917243.42
#Sta/Elev= 30
 -3624.5  160.13 -3474.5  158.35 -3244.5  160.52 -3124.5  156.15 -2944.5  159.28
   -54.5  151.05  1715.5  153.26  1885.5  151.17  2125.5  153.28  2325.5  151.04
  2675.5  153.52  3035.5  150.09  3615.5  152.56  3835.5  149.12  4115.5  154.69
  4265.5  149.39  4365.5  141.74  4575.5  152.12  4895.5   154.3  4925.5  153.76
 4998.71  141.01  5071.8  153.29  5111.8  153.73  5601.8  151.62  5711.8  148.22
  6001.8  151.82  6741.8  151.21  6841.8  148.64  6891.8  153.63  6951.8   154.8
#Mann= 3 ,-1 , 0
 -3624.5     .99       0  4895.5     .04       0  5111.8     .99       0
Levee=0,,,-1,5270.25,151.36,,
#XS Ineff= 2 , 0
       0    4844   151.6    5154       0   151.6
Permanent Ineff=
       F       F
#Block Obstruct= 1 ,-1
 4209.78 4556.96   151.3
Bank Sta=4925.5,5071.8
XS Rating Curve= 0
Exp/Cntr=.3,.1

Type RM Length L Ch R = 1 ,16594   ,156.56,160,163.69
BEGIN DESCRIPTION:
Added channel cross section
END DESCRIPTION:
XS GIS Cut Line= 6
   3014529.8757613926747.9720319 3011659.114254913920333.7092272
 3011410.466425113918924.0259067 3011399.236122213918817.8023354
 3011387.096091613918767.7962657 3010896.175614613916940.1454147
#Sta/Elev= 30
-3588.18  159.85-3176.84  157.58-2910.72  159.14-2631.76   156.7-1994.14  157.03
-1641.81   154.2   63.76  150.66 2688.36  153.31 3047.02  151.02 3624.86  152.44
 3872.72  149.75 4083.41  152.66  4390.1   152.8  4510.1   150.9 4680.91  153.75
  4940.6  152.61  4998.1  137.94    5024  143.11  5053.3  151.98  5097.7   150.7
  5131.3  154.35 5302.72  150.54 5370.83  152.63 5516.78  151.88 5697.18  148.25
 6223.85  151.63 6616.34  149.83 6801.22  150.88 6849.87  148.74 6998.36  153.94
#Mann= 4 ,-1 , 0
-3588.18     .99       0  4940.6     .04       0  5053.3     .99       0
 6998.36     .99       0
Levee=0,,,-1,5228.517,150.7947,,
Bank Sta=4940.6,5053.3
XS Rating Curve= 0
Exp/Cntr=.3,.1

Type RM Length L Ch R = 1 ,16434   ,420.75,430,439.91
BEGIN DESCRIPTION:
Added channel cross section
END DESCRIPTION:
XS GIS Cut Line= 6
 3014526.121443713926738.3276806 3011709.304654213920316.4304289
  3011557.17453913918882.5165983 3011554.655830313918774.5025719
 3011545.296698813918723.6843108 3011160.641107413916861.7227283
#Sta/Elev= 30
 -3579.1  159.78 -3278.4  159.84-3168.14   157.1-2987.72  159.47-2623.57  156.66
-2005.42  157.05-1634.55  154.11   69.43   150.5 2691.57  153.26 3186.72  150.88
  3627.2  152.41 3874.83  149.88 4025.18   152.3  4510.1   150.9 4656.66  153.56
 4885.29  151.42  4938.6  153.09  4971.8  142.81    4998  138.38    5040   143.1
  5073.6  151.48    5132  153.97 5300.94  149.67 5369.59  152.42 5698.53  148.22
 5997.27   148.7 6166.91  151.59  6811.3  150.83 6860.34   148.7    7010  153.73
#Mann= 4 ,-1 , 0
 -3579.1     .99       0  4938.6     .04       0  5073.6     .99       0
    7010     .99       0
Levee=0,,,-1,5192,150.3,,
Bank Sta=4938.6,5073.6
XS Rating Curve= 0
Exp/Cntr=.3,.1

Type RM Length L Ch R = 1 ,16004   ,737.64,750,759.89
BEGIN DESCRIPTION:
Cross Section K145-00-00-X6 (updated with channel survey for Cypress Rosehill)
END DESCRIPTION:
XS GIS Cut Line= 5
 3014544.790142313926702.8499407        3011850.     13920235.35
      3011945.88     13918754.75       3011966.2     13918643.89
        3011850.     13916654.62
#Sta/Elev= 30
 -3556.4   159.6 -3256.4   159.9 -3156.4   155.9 -2966.4   159.9 -1566.4   153.7
  -236.4   153.4    83.6   150.1  2743.6   153.3  3193.6   150.2  3343.6   153.1
  3470.1   150.3  4030.1   152.1  4140.1   149.5  4250.1   152.7  4861.9   152.7
  4888.2  149.98  4933.9  152.84  4954.2   144.5  4997.6  137.72  5068.9  150.93
  5105.7  149.41  5128.6  153.07  5296.5   147.5  5366.5   151.9  5516.5   151.5
  5586.5   147.4  6006.5   147.2  6116.5   151.6  6886.5   148.6  7039.1   153.2
#Mann= 3 ,-1 , 0
 -3556.4     .99       0  4933.9     .04       0  5068.9     .99       0
Levee=0,,,-1,5192,150.3,,
Bank Sta=4933.9,5068.9
XS Rating Curve= 0
Exp/Cntr=.3,.1

Type RM Length L Ch R = 1 ,15254   ,157.37,160,162.11
BEGIN DESCRIPTION:
Added channel cross section
END DESCRIPTION:
XS GIS Cut Line= 5
      3014867.12      13927450.1      3012300.57     13920308.77
      3012670.71     13919059.05      3012722.39       13918949.
       3012508.9     13916428.56
#Sta/Elev= 30
 -3952.3  166.46 -2852.3  159.78 -2762.3  155.75 -2572.3  160.12 -2422.3  153.34
 -1762.3  157.39 -1222.3  153.21   657.7  150.43  1837.7  153.37  2637.7  150.73
  2797.7  153.74    4934  151.79  4992.1  136.96  5041.3     143    5069  151.33
  5181.3  150.44  5231.3  155.12  5321.3  151.01  5701.3  151.06  5851.3  147.17
  5911.3  150.44  6001.3  147.54  6331.3  151.06  6451.3  147.58  6511.3  150.17
  7161.3  145.86  7401.3     148  7461.3  160.59  7561.3  160.86  7590.7  154.18
#Mann= 3 ,-1 , 0
 -3952.3     .99       0    4934     .04       0    5069     .99       0
Levee=0,,,-1,5084.12,150.02,,
Bank Sta=4934,5069
XS Rating Curve= 0
Exp/Cntr=.5,.3

Type RM Length L Ch R = 1 ,15094   ,20,20,20
BEGIN DESCRIPTION:
S5-1_PL-US - XS3 (updated with channel survey)
END DESCRIPTION:
XS GIS Cut Line= 5
      3014903.99     13927445.67      3012390.96     13920362.33
      3012761.11     13919112.62      3012812.78     13919002.57
       3012599.3     13916482.13
#Sta/Elev= 30
 -3890.8  166.56 -2810.8  159.78 -2710.8  155.79 -2550.8  159.31 -2010.8  155.34
  1289.2  149.97  1889.2  153.69  2059.2   151.1  2859.2  154.13  3019.2  151.15
  3159.2   153.8  3609.2  150.67  3765.1  153.44    4932  151.81    4991  136.97
    5050  151.69  5079.6  152.28  5290.1  148.66  5340.1  153.16  5400.1  150.17
  5910.1  150.35  5960.1  146.85  6170.1  151.25  6580.1  147.28  6640.1  150.22
  7310.1  150.38  7420.1  147.08  7470.1  148.72  7520.1  161.96  7579.5  163.78
#Mann= 3 ,-1 , 0
 -3890.8     .99       0    4932     .04       0  5079.6     .99       0
Levee=0,,,-1,5110,150,,
#XS Ineff= 2 , 0
       0    4932  146.86  5079.6       0  146.86
Permanent Ineff=
       F       F
Bank Sta=4932,5079.6
XS Rating Curve= 0
Exp/Cntr=.5,.3

Type RM Length L Ch R = 3 ,15084   ,,,
BEGIN DESCRIPTION:
PL1_K145-00-00-S5-1
END DESCRIPTION:
Bridge Culvert--1,0,-1,-1, 0
Deck Dist Width WeirC Skew NumUp NumDn MinLoCord MaxHiCord MaxSubmerge Is_Ogee
10,1,2.6,0, 9, 9, , , .95, 0, ,,,
  4938.2  4938.3 4938.41  4938.6  4942.6  5077.1 5079.39  5079.5  5079.6
  150.51  150.51  150.59  150.66  153.59  153.53  152.36  152.28  152.28
  150.51  150.48  150.44  150.41  152.92  152.86  152.27  152.27  152.28
  4938.2  4938.3 4938.41  4938.6  4942.6  5077.1 5079.39  5079.5  5079.6
  150.51  150.51  150.59  150.66  153.59  153.53  152.36  152.28  152.28
  150.51  150.48  150.44  150.41  152.92  152.86  152.27  152.27  152.28
Pier Skew, UpSta & Num, DnSta & Num=  ,4945.2, 2 ,4945.2, 2 , 0 , 0 , 0 ,,
     1.3     1.3
  147.05  153.92
     1.3     1.3
  147.05  153.92
Pier Skew, UpSta & Num, DnSta & Num=  ,4960.2, 2 ,4960.2, 2 , 0 , 0 , 0 ,,
     1.3     1.3
  142.92  153.91
     1.3     1.3
  142.92  153.91
Pier Skew, UpSta & Num, DnSta & Num=  ,4980.6, 2 ,4980.6, 2 , 0 , 0 , 0 ,,
     1.3     1.3
  136.91   153.9
     1.3     1.3
  136.91   153.9
Pier Skew, UpSta & Num, DnSta & Num=  ,5000.6, 2 ,5000.6, 2 , 0 , 0 , 0 ,,
     1.3     1.3
   138.6  153.89
     1.3     1.3
   138.6  153.89
Pier Skew, UpSta & Num, DnSta & Num=  ,5020.6, 2 ,5020.6, 2 , 0 , 0 , 0 ,,
     1.3     1.3
  142.68  153.89
     1.3     1.3
  142.68  153.89
Pier Skew, UpSta & Num, DnSta & Num=  ,5039.6, 2 ,5039.6, 2 , 0 , 0 , 0 ,,
     1.3     1.3
  147.92  153.88
     1.3     1.3
  147.92  153.88
BR Coef= 1 , 1 , 1 ,1.25, 0 ,,,.8,0,2,0,
WSPro=,,,, 1 ,,,, 0 ,,,, 0 ,,,,-1 ,-1 ,-1 , 0 , 0 , 0 , 0 , 0
BR U #Sta/Elev= 30
 -3890.8  166.56 -2810.8  159.78 -2710.8  155.79 -2550.8  159.31 -2010.8  155.34
  1289.2  149.97  1889.2  153.69  2059.2   151.1  2859.2  154.13  3019.2  151.15
  3159.2   153.8  3609.2  150.67  3765.1  153.44    4932  151.81    4991  136.97
    5050  151.69  5079.6  152.28  5290.1  148.66  5340.1  153.16  5400.1  150.17
  5910.1  150.35  5960.1  146.85  6170.1  151.25  6580.1  147.28  6640.1  150.22
  7310.1  150.38  7420.1  147.08  7470.1  148.72  7520.1  161.96  7579.5  163.78
BR U #Mann= 3
 -3890.8     .99    4932     .04  5079.6     .99
BR U Banks=4932,5079.6
BR D #Sta/Elev= 30
 -3890.8  166.53 -2810.8  159.75 -2710.8  155.76 -2550.8  159.28 -2010.8  155.31
  1289.2  149.94  1889.2  153.66  2059.2  151.07  2859.2   154.1  3019.2  151.12
  3159.2  153.77  3609.2  150.64  3765.1  153.41    4932  151.81    4991  136.97
    5050  151.69  5079.6  152.28  5290.1  148.63  5340.1  153.13  5400.1  150.14
  5910.1  150.32  5960.1  146.82  6170.1  151.22  6580.1  147.25  6640.1  150.19
  7310.1  150.35  7420.1  147.05  7470.1  148.69  7520.1  161.93  7579.5  163.75
BR D #Mann= 3
 -3890.8     .99    4932     .04  5079.6     .99
BR D Banks=4932,5079.6
BC Design=,, 0 ,, 0 ,,,,,,
BC HTab HWMax=166.56

Type RM Length L Ch R = 1 ,15074   ,104.81,100,96.39
BEGIN DESCRIPTION:
S5-1_PL-DS - XS2 (updated with channel survey)
END DESCRIPTION:
XS GIS Cut Line= 5
      3014922.83     13927438.98      3012411.99     13920361.78
      3012779.85     13919119.75      3012833.16     13919006.22
      3012619.23     13916480.44
#Sta/Elev= 30
 -3890.8  166.53 -2810.8  159.75 -2710.8  155.76 -2550.8  159.28 -2010.8  155.31
  1289.2  149.94  1889.2  153.66  2059.2  151.07  2859.2   154.1  3019.2  151.12
  3159.2  153.77  3609.2  150.64  3765.1  153.41    4932  151.81    4991  136.97
    5050  151.69  5079.6  152.28  5290.1  148.63  5340.1  153.13  5400.1  150.14
  5910.1  150.32  5960.1  146.82  6170.1  151.22  6580.1  147.25  6640.1  150.19
  7310.1  150.35  7420.1  147.05  7470.1  148.69  7520.1  161.93  7579.5  163.75
#Mann= 3 ,-1 , 0
 -3890.8     .99       0    4932     .04       0  5079.6     .99       0
Levee=0,,,-1,5110,150,,
#XS Ineff= 2 , 0
       0    4932  146.86  5079.6       0  146.86
Permanent Ineff=
       F       F
Bank Sta=4932,5079.6
XS Rating Curve= 0
Exp/Cntr=.5,.3

Type RM Length L Ch R = 1 ,14974   ,313.38,299,288.22
BEGIN DESCRIPTION:
S5-1_PL-DS - XS1 (updated with channel survey)
END DESCRIPTION:
XS GIS Cut Line= 5
       3014925.2      13927437.5      3012507.96     13920401.95
      3012875.83     13919159.92      3012929.14     13919046.39
       3012715.2     13916520.61
#Sta/Elev= 30
 -3798.6  166.47 -2628.6  155.71 -2478.6  159.85 -2348.6  158.07 -2298.6  153.17
 -2078.6  152.66 -1588.6  156.54 -1348.6  156.22 -1308.6  152.04 -1268.6  155.53
   451.4  150.88  2931.4  154.03  3720.6  150.37  4680.6  152.44  4780.6  149.35
  4910.6  152.43  4930.6  151.36 4992.93  137.46    5056  151.11  5081.4  151.75
  5351.4   149.3  5381.4  156.08  5421.4  150.03  5601.4  147.05  5841.4  150.57
  6651.4  147.37  7211.4  151.17  7481.4  147.16  7541.4  148.76  7596.2  164.09
#Mann= 3 ,-1 , 0
 -3798.6     .99       0  4910.6     .04       0  5081.4     .99       0
Levee=0,,,-1,5106.92,150.01,,
Bank Sta=4930.6,5056
XS Rating Curve= 0
Exp/Cntr=.3,.1

Type RM Length L Ch R = 1 ,14675   ,104.81,100,96.39
BEGIN DESCRIPTION:
S5A_PL-DS - XS4 (updated with channel survey)
END DESCRIPTION:
XS GIS Cut Line= 5
      3014897.98      13927352.5      3013045.25     13921017.59
      3013184.38     13919263.56      3013186.13     13919145.59
      3013028.88     13916412.23
#Sta/Elev= 30
   -3429   166.2   -2359  155.97   -2139  159.44   -1999  152.15   -1829     152
   -1759  155.91   -1109  156.65   -1059  150.94   -1029  155.42    2461  151.89
    2591  149.36    2721  153.35    2841  150.91  3491.3  153.99  3741.3  150.48
  4901.3  152.01  4930.9  150.77 4997.31  136.43  5058.9  151.15  5088.9  151.71
  5348.9  150.36  5388.9  158.71  5448.9  151.65  5658.9  147.69  7068.9  149.45
  7128.9  150.95  7168.9  160.91  7248.9  168.44  7288.9  166.19  7328.9  172.09
#Mann= 3 ,-1 , 0
   -3429     .99       0  4901.3     .04       0  5088.9     .99       0
Levee=0,,,-1,5401.69,150.79,,
Bank Sta=4930.9,5058.9
XS Rating Curve= 0
Exp/Cntr=.5,.3

Type RM Length L Ch R = 1 ,14575   ,14,15,15
BEGIN DESCRIPTION:
S5A_PL-DS - XS3 (updated with channel survey)
END DESCRIPTION:
XS GIS Cut Line= 5
      3014908.18     13927357.75       3013140.7      13921025.6
      3013279.83     13919271.57      3013281.58     13919153.61
      3013124.32     13916420.25
#Sta/Elev= 30
 -3398.2  166.35 -2398.2  159.16 -2338.2  156.43 -2088.2  159.17 -1688.2   155.1
 -1078.2  156.56  -788.2  153.55  -568.2  155.28   731.8  150.83  2781.8  152.14
  2891.8  149.59  3001.8  152.88    3516  154.24    3556  150.83    4356  153.07
    4396  149.98    4656  152.43 4944.37  150.44 4998.77  136.09 5052.07  150.59
  5193.5  150.65  5343.5  155.88  5523.5  150.74  6283.5  150.56  6443.5  147.76
  7343.5  151.06  7683.5  148.11  7723.5  148.92  7773.5  166.01  7791.4  168.67
#Mann= 3 ,-1 , 0
 -3398.2     .99       0 4944.37     .04       0 5052.07     .99       0
Levee=0,,,-1,5174,150,,
#XS Ineff= 2 , 0
       0 4944.37  147.72 5052.07       0  147.72
Permanent Ineff=
       F       F
Bank Sta=4944.37,5052.07
XS Rating Curve= 0
Exp/Cntr=.5,.3

Type RM Length L Ch R = 3 ,14565   ,,,
BEGIN DESCRIPTION:
PL1_K145-00-00-S5A
END DESCRIPTION:
Bridge Culvert--1,0,-1,-1, 0
Deck Dist Width WeirC Skew NumUp NumDn MinLoCord MaxHiCord MaxSubmerge Is_Ogee
10,1,2.6,0, 60, 60, , , .95, 0, ,,,
 -3398.2 -3078.2 -2708.2 -2648.2 -2398.2 -2338.2 -2288.2 -2088.2 -1688.2 -1078.2
 -1008.2  -808.2  -788.2  -768.2  -738.2  -568.2   391.8   731.8  1441.8  1631.8
  2641.8  2711.8  2781.8  2861.8  2891.8  2971.8  3001.8    3516    3556    3596
    4126    4356    4396    4526    4556    4636    4656 4896.27 4944.97 5050.17
 5058.07  5193.5  5343.5  5373.5  5403.5  5493.5  5523.5  6283.5  6443.5  6483.5
  7123.5  7173.5  7343.5  7423.5  7683.5  7723.5  7733.5  7743.5  7773.5  7791.4
  166.31  164.51  160.07  161.08  159.12  156.39  158.42  159.13  155.06  156.52
  154.74  154.94  153.51  154.91   153.9  155.24  153.17  150.79  152.37  150.81
  151.26   150.3   152.1  151.65  149.55  150.92  152.84   154.2  150.79  152.84
  151.83  153.03  149.94  152.23  150.95  150.91  152.39  152.33  151.18  150.86
  152.05  150.61  155.84  155.37  152.53  152.05   150.7  150.52  147.72  149.93
   150.6   149.3  151.02  149.13  148.07  148.88  152.06  157.05  165.97  168.63
  166.31  164.51  160.07  161.08  159.12  156.39  158.42  159.13  155.06  156.52
  154.74  154.94  153.51  154.91   153.9  155.24  153.17  150.79  152.37  150.81
  151.26   150.3   152.1  151.65  149.55  150.92  152.84   154.2  150.79  152.84
  151.83  153.03  149.94  152.23  150.95  150.91  152.39  152.33  150.18  149.81
  152.05  150.61  155.84  155.37  152.53  152.05   150.7  150.52  147.72  149.93
   150.6   149.3  151.02  149.13  148.07  148.88  152.06  157.05  165.97  168.63
 -3398.2 -3078.2 -2708.2 -2648.2 -2398.2 -2338.2 -2288.2 -2088.2 -1688.2 -1078.2
 -1008.2  -808.2  -788.2  -768.2  -738.2  -568.2   391.8   731.8  1441.8  1631.8
  2641.8  2711.8  2781.8  2861.8  2891.8  2971.8  3001.8    3516    3556    3596
    4126    4356    4396    4526    4556    4636    4656 4896.27 4944.97 5050.17
 5058.07  5193.5  5343.5  5373.5  5403.5  5493.5  5523.5  6283.5  6443.5  6483.5
  7123.5  7173.5  7343.5  7423.5  7683.5  7723.5  7733.5  7743.5  7773.5  7791.4
  166.31  164.51  160.07  161.08  159.12  156.39  158.42  159.13  155.06  156.52
  154.74  154.94  153.51  154.91   153.9  155.24  153.17  150.79  152.37  150.81
  151.26   150.3   152.1  151.65  149.55  150.92  152.84   154.2  150.79  152.84
  151.83  153.03  149.94  152.23  150.95  150.91  152.39  152.33  151.18  150.86
  152.05  150.61  155.84  155.37  152.53  152.05   150.7  150.52  147.72  149.93
   150.6   149.3  151.02  149.13  148.07  148.88  152.06  157.05  165.97  168.63
  166.31  164.51  160.07  161.08  159.12  156.39  158.42  159.13  155.06  156.52
  154.74  154.94  153.51  154.91   153.9  155.24  153.17  150.79  152.37  150.81
  151.26   150.3   152.1  151.65  149.55  150.92  152.84   154.2  150.79  152.84
  151.83  153.03  149.94  152.23  150.95  150.91  152.39  152.33  150.18  149.81
  152.05  150.61  155.84  155.37  152.53  152.05   150.7  150.52  147.72  149.93
   150.6   149.3  151.02  149.13  148.07  148.88  152.06  157.05  165.97  168.63
Pier Skew, UpSta & Num, DnSta & Num=  ,4952, 2 ,4952, 2 , 0 , 0 , 0 ,,
     1.3     1.3
  146.14  151.16
     1.3     1.3
  146.14  151.16
Pier Skew, UpSta & Num, DnSta & Num=  ,4991.8, 2 ,4991.8, 2 , 0 , 0 , 0 ,,
     1.3     1.3
  137.41  151.04
     1.3     1.3
  137.41  151.04
Pier Skew, UpSta & Num, DnSta & Num=  ,5030.8, 2 ,5030.8, 2 , 0 , 0 , 0 ,,
     1.3     1.3
  142.81  150.92
     1.3     1.3
  142.81  150.92
BR Coef= 1 , 1 , 1 ,1.25, 0 ,,,.8,0,2,0,
WSPro=,,,, 1 ,,,, 0 ,,,, 0 ,,,,-1 ,-1 ,-1 , 0 , 0 , 0 , 0 , 0
BR U #Sta/Elev= 198
 -3398.2  166.31 -3098.2  164.31 -3078.2  164.51 -2868.2  161.78 -2838.2  161.05
 -2708.2  160.07 -2668.2   160.2 -2648.2  161.08 -2398.2  159.12 -2368.2     158
 -2358.2  156.77 -2338.2  156.39 -2318.2     157 -2288.2  158.42 -2088.2  159.13
 -2058.2  158.55 -1748.2  155.72 -1728.2  155.71 -1688.2  155.06 -1668.2   155.7
 -1648.2  155.64 -1638.2  155.93 -1358.2  155.57 -1338.2  156.14 -1198.2  155.87
 -1078.2  156.52 -1008.2  154.74  -998.2  155.05  -888.2  154.13  -808.2  154.94
  -798.2   154.6  -788.2  153.51  -778.2  153.54  -768.2  154.91  -758.2  154.77
  -748.2   154.1  -738.2   153.9  -698.2  154.65  -608.2  154.94  -588.2  154.51
  -568.2  155.24  -438.2  154.21  -348.2  154.77  -208.2  153.76  -188.2   154.2
    41.8  153.13    51.8  153.54    81.8  152.98   251.8  153.36   311.8  153.13
   331.8  153.33   391.8  153.17   491.8   151.9   591.8  152.21   731.8  150.79
   761.8  151.03  1051.8  151.63  1401.8  151.44  1441.8  152.37  1541.8  151.19
  1631.8  150.81  2631.8  150.93  2641.8  151.26  2671.8  150.39  2711.8   150.3
  2747.3  151.21  2781.8   152.1  2861.8  151.65  2881.8  150.69  2891.8  149.55
  2931.8  149.73  2971.8  150.92  3001.8  152.84  3081.8  153.38  3101.8  153.01
  3141.8  153.47    3176  152.94    3326  153.49    3356  153.08    3396  153.96
    3456  153.54    3516   154.2    3526  153.83    3536  152.93    3546  151.47
    3556  150.79  3558.3  150.87    3566  151.12    3576   152.3    3596  152.84
    3616   152.6    3676   152.6    3706  152.29    3926  152.39    3946  151.98
    4126  151.83    4186  152.31    4226  152.78    4356  153.03    4366  152.74
    4386  150.54    4396  149.94    4456  150.12    4506  151.38    4526  152.23
    4546  151.65    4556  150.95    4636  150.91    4656  152.39    4786  151.82
 4896.27  152.33 4929.97  151.61  4936.4   151.3 4939.27  151.17 4941.27  151.07
  4944.2  150.44 4944.37   150.4 4944.88  150.19 4944.97  150.16 4951.97  147.32
 4964.17  143.92 4980.17  139.83 4990.17  138.33 4991.77  138.74 4993.37  137.93
 4994.07  137.37 4998.77  136.05 5003.97  136.78 5006.57  138.09 5008.47  138.63
 5024.77  141.86 5030.77  144.05 5043.47  147.22 5050.06  149.77 5050.17  149.81
 5052.07  150.55 5054.27   151.1  5054.5  151.16 5058.07  152.05 5084.37  151.96
 5111.37  151.56  5173.5  150.55  5193.5  150.61  5203.5  151.32  5223.5  151.86
  5233.5  152.64  5283.5  153.68  5343.5  155.84  5363.5  155.82  5373.5  155.37
  5383.5  154.01  5393.5  153.53  5403.5  152.53  5413.5   153.2  5463.5  151.76
  5493.5  152.05  5523.5   150.7  5613.5  150.59  5653.5  151.24  5693.5  150.61
  5783.5  151.38  5813.5  150.56  5993.5  150.71  6013.5  150.09  6063.5  150.25
  6073.5  149.82  6153.5  149.75  6183.5  150.12  6283.5  150.52  6303.5  150.01
  6333.5  150.16  6363.5  149.57  6393.5  147.83  6423.5  148.54  6443.5  147.72
  6453.5   147.8  6463.5  149.07  6483.5  149.93  6753.5  150.27  6783.5  149.51
  6833.5   150.2  6903.5  149.91  6953.5  149.98  6963.5  149.64  7053.5   150.4
  7123.5   150.6  7173.5   149.3  7313.5  149.89  7343.5  151.02  7423.5  149.13
  7473.5   149.8  7613.5  148.43  7683.5  148.07  7723.5  148.88  7733.5  152.06
  7743.5  157.05  7773.5  165.97  7791.4  168.63
BR U #Mann= 3
 -3398.2     .99 4944.37     .04 5052.07     .99
BR U Banks=4944.37,5052.07
BR D #Sta/Elev= 198
 -3398.2  166.31 -3098.2  164.31 -3078.2  164.51 -2868.2  161.78 -2838.2  161.05
 -2708.2  160.07 -2668.2   160.2 -2648.2  161.08 -2398.2  159.12 -2368.2     158
 -2358.2  156.77 -2338.2  156.39 -2318.2     157 -2288.2  158.42 -2088.2  159.13
 -2058.2  158.55 -1748.2  155.72 -1728.2  155.71 -1688.2  155.06 -1668.2   155.7
 -1648.2  155.64 -1638.2  155.93 -1358.2  155.57 -1338.2  156.14 -1198.2  155.87
 -1078.2  156.52 -1008.2  154.74  -998.2  155.05  -888.2  154.13  -808.2  154.94
  -798.2   154.6  -788.2  153.51  -778.2  153.54  -768.2  154.91  -758.2  154.77
  -748.2   154.1  -738.2   153.9  -698.2  154.65  -608.2  154.94  -588.2  154.51
  -568.2  155.24  -438.2  154.21  -348.2  154.77  -208.2  153.76  -188.2   154.2
    41.8  153.13    51.8  153.54    81.8  152.98   251.8  153.36   311.8  153.13
   331.8  153.33   391.8  153.17   491.8   151.9   591.8  152.21   731.8  150.79
   761.8  151.03  1051.8  151.63  1401.8  151.44  1441.8  152.37  1541.8  151.19
  1631.8  150.81  2631.8  150.93  2641.8  151.26  2671.8  150.39  2711.8   150.3
  2747.3  151.21  2781.8   152.1  2861.8  151.65  2881.8  150.69  2891.8  149.55
  2931.8  149.73  2971.8  150.92  3001.8  152.84  3081.8  153.38  3101.8  153.01
  3141.8  153.47    3176  152.94    3326  153.49    3356  153.08    3396  153.96
    3456  153.54    3516   154.2    3526  153.83    3536  152.93    3546  151.47
    3556  150.79  3558.3  150.87    3566  151.12    3576   152.3    3596  152.84
    3616   152.6    3676   152.6    3706  152.29    3926  152.39    3946  151.98
    4126  151.83    4186  152.31    4226  152.78    4356  153.03    4366  152.74
    4386  150.54    4396  149.94    4456  150.12    4506  151.38    4526  152.23
    4546  151.65    4556  150.95    4636  150.91    4656  152.39    4786  151.82
 4896.27  152.33 4929.97  151.61  4936.4   151.3 4939.27  151.17 4941.27  151.07
  4944.2  150.44 4944.37   150.4 4944.88  150.19 4944.97  150.16 4951.97  147.32
 4964.17  143.92 4980.17  139.83 4990.17  138.33 4991.77  138.74 4993.37  137.93
 4994.07  137.37 4998.77  136.05 5003.97  136.78 5006.57  138.09 5008.47  138.63
 5024.77  141.86 5030.77  144.05 5043.47  147.22 5050.06  149.77 5050.17  149.81
 5052.07  150.55 5054.27   151.1  5054.5  151.16 5058.07  152.05 5084.37  151.96
 5111.37  151.56  5173.5  150.55  5193.5  150.61  5203.5  151.32  5223.5  151.86
  5233.5  152.64  5283.5  153.68  5343.5  155.84  5363.5  155.82  5373.5  155.37
  5383.5  154.01  5393.5  153.53  5403.5  152.53  5413.5   153.2  5463.5  151.76
  5493.5  152.05  5523.5   150.7  5613.5  150.59  5653.5  151.24  5693.5  150.61
  5783.5  151.38  5813.5  150.56  5993.5  150.71  6013.5  150.09  6063.5  150.25
  6073.5  149.82  6153.5  149.75  6183.5  150.12  6283.5  150.52  6303.5  150.01
  6333.5  150.16  6363.5  149.57  6393.5  147.83  6423.5  148.54  6443.5  147.72
  6453.5   147.8  6463.5  149.07  6483.5  149.93  6753.5  150.27  6783.5  149.51
  6833.5   150.2  6903.5  149.91  6953.5  149.98  6963.5  149.64  7053.5   150.4
  7123.5   150.6  7173.5   149.3  7313.5  149.89  7343.5  151.02  7423.5  149.13
  7473.5   149.8  7613.5  148.43  7683.5  148.07  7723.5  148.88  7733.5  152.06
  7743.5  157.05  7773.5  165.97  7791.4  168.63
BR D #Mann= 3
 -3398.2     .99 4944.37     .04 5052.07     .99
BR D Banks=4944.37,5052.07
BC Design=,, 0 ,, 0 ,,,,,,
BC HTab HWMax=168.67

Type RM Length L Ch R = 1 ,14560   ,104,105,106
BEGIN DESCRIPTION:
S5_CYPRESS ROSEHILL-DS - XS3  **SEE NOTE**
The right end of this XS stops under an overpass.  This XS cannot be extended to high ground.  This is a spill to the main stem of Cypress unless a levee is possible at sta 5700.
END DESCRIPTION:
XS GIS Cut Line= 6
      3014967.26     13927422.85      3013206.48     13921030.39
      3013318.18     13919271.48      3013321.45     13919155.81
      3013323.21     13918893.01      3013229.07     13916416.98
#Sta/Elev= 30
 -3452.5   166.6 -2472.5     160 -2332.5   156.6 -2142.5   159.8 -1702.5   154.7
 -1282.5   156.7  -722.5   153.3  -362.5   155.6    27.5   152.8  2847.5   151.5
  2917.5   149.6  2977.5   152.3  3147.5     149    3178   151.5    3388     153
    3528   152.8    3578   148.5    3618   152.1    3778   152.5    3828   150.6
    4638   151.1  4952.2  150.85  4999.4  135.51    5011  135.51  5060.6  151.13
    7479   150.1    7559   148.4    7599   150.3    7689   147.5  7796.8   148.4
#Mann= 4 ,-1 , 0
 -3452.5     .99       0    4638      .1       0  4952.2     .04       0
  5060.6     .99       0
Levee=-1,4626,150,-1,5282,150,,
#XS Ineff= 2 , 0
       0  4952.2   147.5  5060.6       0   147.5
Permanent Ineff=
       F       F
Bank Sta=4952.2,5060.6
XS Rating Curve= 0
Exp/Cntr=.5,.3

Type RM Length L Ch R = 3 ,14555   ,,,
BEGIN DESCRIPTION:
CYPRESS-ROSEHILL BRIDGE
Structure ID: K145-00-00-S5
END DESCRIPTION:
Bridge Culvert--1,0,-1,-1, 0
Deck Dist Width WeirC Skew NumUp NumDn MinLoCord MaxHiCord MaxSubmerge Is_Ogee
5,94,2.6,0, 40, 40, , , .95, 0, ,,,
    3528  3611.9  3717.9  3817.9  3917.9  4015.9  4120.9  4225.9  4752.9  4831.9
  4881.9  4960.9  5048.9  5081.9  5166.9  5294.9  5396.9  5497.9  5596.9  5699.9
  5791.9  5895.9  6102.9  6202.9  6301.9  6401.9  6502.9  6531.9  6602.9  6697.9
  6801.9  6889.9  6917.9  7013.9  7110.9  7208.9  7306.9  7407.9  7505.9    7599
   152.8  152.62  152.74  152.88  152.85  152.83  152.64  152.19  151.51  151.63
  151.83  152.87   152.6  152.43  152.01  151.99  152.17  152.29  152.26  152.15
  152.05  152.03  151.71   151.3  151.16  151.38  151.35  151.23  151.21  151.04
  150.93  150.91  150.73  150.76  150.81  150.78  150.74  150.66  150.52   150.3
                                                                                
          150.28  150.01
                                                                                
                                                                                
    3528  3611.9  3717.9  3817.9  3917.9  4015.9  4120.9  4225.9  4752.9  4831.9
  4881.9  4960.9  5048.9  5081.9  5166.9  5294.9  5396.9  5497.9  5596.9  5699.9
  5791.9  5895.9  6102.9  6202.9  6301.9  6401.9  6502.9  6531.9  6602.9  6697.9
  6801.9  6889.9  6917.9  7013.9  7110.9  7208.9  7306.9  7407.9  7505.9    7599
   152.8  152.62  152.74  152.88  152.85  152.83  152.64  152.19  151.51  151.63
  151.83  152.87   152.6  152.43  152.01  151.99  152.17  152.29  152.26  152.15
  152.05  152.03  151.71   151.3  151.16  151.38  151.35  151.23  151.21  151.04
  150.93  150.91  150.73  150.76  150.81  150.78  150.74  150.66  150.52   150.3
                                                                                
          150.28  150.01
                                                                                
                                                                                
Pier Skew, UpSta & Num, DnSta & Num=  ,4989.9, 2 ,4989.9, 2 , 0 , 0 , 0 ,,
    1.35    1.35
  137.17   151.8
    1.35    1.35
  137.17   151.8
Pier Skew, UpSta & Num, DnSta & Num=  ,5019.9, 2 ,5019.9, 2 , 0 , 0 , 0 ,,
    1.35    1.35
  137.16  151.86
    1.35    1.35
  137.16  151.86
BR Coef= 1 , 1 , 1 ,1.25, 0 ,,,.8,0,2,0,
WSPro=,,,, 1 ,,,, 0 ,,,, 0 ,,,,-1 ,-1 ,-1 , 0 , 0 , 0 , 0 , 0
BR U #Sta/Elev= 148
 -3452.5   166.6 -3022.5   163.9 -2962.5   163.8 -2932.5   163.3 -2912.5   163.6
 -2702.5   160.5 -2682.5   160.9 -2652.5   160.9 -2632.5   161.4 -2492.5   159.7
 -2472.5     160 -2372.5   158.5 -2342.5   156.8 -2332.5   156.6 -2322.5     157
 -2312.5   157.9 -2222.5     160 -2142.5   159.8 -2122.5     159 -2082.5   159.3
 -2042.5   158.2 -2032.5   157.5 -1732.5   156.4 -1722.5   156.1 -1702.5   154.7
 -1682.5   154.8 -1512.5   155.4 -1502.5   155.1 -1422.5     156 -1402.5   156.1
 -1362.5   155.6 -1282.5   156.7 -1132.5   155.9 -1072.5   156.2 -1002.5   155.6
  -962.5   154.1  -832.5     155  -762.5     154  -742.5     155  -722.5   153.3
  -712.5   154.4  -702.5   154.9  -632.5   154.1  -612.5   154.7  -552.5   154.7
  -522.5   153.9  -382.5   154.5  -362.5   155.6  -302.5   154.1   -32.5   153.3
    27.5   152.8   247.5   152.5   367.5     153   387.5   152.8   477.5   153.1
   507.5   152.4   527.5   152.5   547.5   151.9   647.5   151.9   677.5   151.8
  1017.5   151.4  1037.5     151  1057.5   151.9  1127.5   151.5  1467.5   151.3
  1477.5   151.7  2157.5     151  2167.5   150.6  2187.5   151.1  2817.5     151
  2847.5   151.5  2887.5     151  2917.5   149.6  2977.5   152.3  3087.5   151.4
  3127.5   149.1  3147.5     149  3167.5   150.3  3177.5   151.4    3178   151.5
    3218   151.4    3258   151.2    3288   152.4    3388     153    3408   152.5
    3468   152.1    3498   152.7    3528   152.8    3538   152.3    3558   149.4
    3578   148.5    3588   148.6    3618   152.1    3748   151.7    3778   152.5
    3808     152    3828   150.6    3858   151.7    3928   151.3    3938     151
    3958   151.7    4148   150.4    4448   149.6    4498   149.9    4518   151.1
    4638   151.1  4925.9   150.6  4952.2  150.85  4960.9  148.35  4999.4  135.51
    5011  135.51  5048.9  148.15  5060.6  151.13  5069.5  151.21  5106.2   151.6
  5166.2   151.3    5709   150.7    5859   150.6    5979   150.6    6129   149.9
    6319   150.5    6349   150.8    6399   149.5    6429   149.9    6449   149.5
    6489   150.1    6689   149.6    6709   149.8    6729   150.7    7039   149.2
    7059   150.3    7209   149.4    7319   149.5    7359   149.3    7389   149.6
    7399   149.4    7429   150.1    7459   149.7    7479   150.1    7559   148.4
    7579   148.9    7599   150.3    7609   150.2    7629   148.6    7669   148.5
    7689   147.5    7699     148  7796.8   148.4
BR U #Mann= 4
 -3452.5     .99    4638      .1  4952.2    .035  5060.6     .99
BR D #Sta/Elev= 148
 -3452.5   166.6 -3022.5   163.9 -2962.5   163.8 -2932.5   163.3 -2912.5   163.6
 -2702.5   160.5 -2682.5   160.9 -2652.5   160.9 -2632.5   161.4 -2492.5   159.7
 -2472.5     160 -2372.5   158.5 -2342.5   156.8 -2332.5   156.6 -2322.5     157
 -2312.5   157.9 -2222.5     160 -2142.5   159.8 -2122.5     159 -2082.5   159.3
 -2042.5   158.2 -2032.5   157.5 -1732.5   156.4 -1722.5   156.1 -1702.5   154.7
 -1682.5   154.8 -1512.5   155.4 -1502.5   155.1 -1422.5     156 -1402.5   156.1
 -1362.5   155.6 -1282.5   156.7 -1132.5   155.9 -1072.5   156.2 -1002.5   155.6
  -962.5   154.1  -832.5     155  -762.5     154  -742.5     155  -722.5   153.3
  -712.5   154.4  -702.5   154.9  -632.5   154.1  -612.5   154.7  -552.5   154.7
  -522.5   153.9  -382.5   154.5  -362.5   155.6  -302.5   154.1   -32.5   153.3
    27.5   152.8   247.5   152.5   367.5     153   387.5   152.8   477.5   153.1
   507.5   152.4   527.5   152.5   547.5   151.9   647.5   151.9   677.5   151.8
  1017.5   151.4  1037.5     151  1057.5   151.9  1127.5   151.5  1467.5   151.3
  1477.5   151.7  2157.5     151  2167.5   150.6  2187.5   151.1  2817.5     151
  2847.5   151.5  2887.5     151  2917.5   149.6  2977.5   152.3  3087.5   151.4
  3127.5   149.1  3147.5     149  3167.5   150.3  3177.5   151.4    3178   151.5
    3218   151.4    3258   151.2    3288   152.4    3388     153    3408   152.5
    3468   152.1    3498   152.7    3528   152.8    3538   152.3    3558   149.4
    3578   148.5    3588   148.6    3618   152.1    3748   151.7    3778   152.5
    3808     152    3828   150.6    3858   151.7    3928   151.3    3938     151
    3958   151.7    4148   150.4    4448   149.6    4498   149.9    4518   151.1
    4638   151.1  4925.9   150.6  4952.2  150.85  4960.9  148.35  4999.4  135.51
    5011  135.51  5048.9  148.15  5060.6  151.13  5069.5  151.21  5106.2   151.6
  5166.2   151.3    5709   150.7    5859   150.6    5979   150.6    6129   149.9
    6319   150.5    6349   150.8    6399   149.5    6429   149.9    6449   149.5
    6489   150.1    6689   149.6    6709   149.8    6729   150.7    7039   149.2
    7059   150.3    7209   149.4    7319   149.5    7359   149.3    7389   149.6
    7399   149.4    7429   150.1    7459   149.7    7479   150.1    7559   148.4
    7579   148.9    7599   150.3    7609   150.2    7629   148.6    7669   148.5
    7689   147.5    7699     148  7796.8   148.4
BR D #Mann= 4
 -3452.5     .99  2977.5      .1  4952.2    .035  5060.6     .99
BC Design=,, 0 ,, 0 ,,,,,,
BC HTab HWMax=166.72
